--- VALLEYFK.prj (project) ---

Proj Title=VALLEYFK
Current Plan=p01
Default Exp/Contr=0,0
English Units
Geom File=g01
Flow File=f01
Plan File=p01
Background Map Layer=Inundation Boundary (P100yr Value_0)
BEGIN DESCRIPTION:
----------MODEL BY WOOD PLC 2022----------
AFH study
Randolph County, WV
HEC-RAS Version: RAS 6.2
Vertical Datum: NAVD88
Projection: NAD 1983 StatePlane West Virginia S FIPS 4702 (US Feet)
Terrain: 1-meter LIDAR (FEMA Region III 3DEP collected 2016-2018)
Land Use: 2019 NLCD
Hydrologic Method:
WV SIR2010-5033 regression equations
Additional Model Notes:
VALLEYFK Lower Reach
Split VALLEYFK at the confluence with MUDLKRN
END DESCRIPTION:
DSS Export Rating Curves= 0
DSS Export Rating Curve Sorted= 0
DSS Export Volume Flow Curves= 0
DXF OffsetX= 0
DXF OffsetY= 0
DXF ScaleX= 0
DXF ScaleY= 0

--- VALLEYFK.p01 (plan) ---

Plan Title=Floodplain
Program Version=6.20
Short Identifier=Floodplain
Geom File=g01
Flow File=f01
Subcritical Flow
K Sum by GR= 0
Std Step Tol= 0.01
Critical Tol= 0.01
Num of Std Step Trials= 20
Max Error Tol= 0.3
Flow Tol Ratio= 0.001
Split Flow NTrial= 30
Split Flow Tol= 0.02
Split Flow Ratio= 0.02
Log Output Level= 0
Friction Slope Method= 1
Unsteady Friction Slope Method= 2
Unsteady Bridges Friction Slope Method= 1
Parabolic Critical Depth
Global Vel Dist= 0 , 0 , 0
Global Log Level= 0
CheckData=True
Encroach Param=-1 ,0,0, 0
Mapping Interval=1HOUR
Computation Time Step Use Courant=        0
Computation Time Step Use Time Series=    0
Computation Time Step Count To Double=0
Computation Time Step Max Doubling=0
Computation Time Step Max Halving=0
Computation Time Step Residence Courant=0
Run HTab= 0
Run UNet= 0
Run Sediment= 0
Run PostProcess= 0
Run WQNet= 0
Run RASMapper=-1
UNET Theta= 0
UNET Theta Warmup= 0
UNET ZTol= 0
UNET ZSATol= 0
UNET MxIter= 0
UNET Max Iter WO Improvement= 0
UNET MaxInSteps= 0
UNET DtIC= 0
UNET DtMin= 0
UNET MaxCRTS= 0
UNET WFStab= 0
UNET SFStab= 0
UNET WFX= 1
UNET SFX= 1
UNET Gravity=32.174
UNET 1D Methodology=Finite Difference
UNET DSS MLevel= 1
UNET Pardiso=0
UNET DZMax Abort= 0
UNET Use Existing IB Tables= 0
UNET Froude Reduction=False
UNET Froude Limit= 0
UNET Froude Power= 0
UNET D1 Cores= 0
UNET WindReference=Eulerian
UNET WindDragFormulation=Hsu (1988)
UNET D2 Coriolis=0
UNET D2 Cores= 0
UNET D2 Theta= 1
UNET D2 Theta Warmup= 1
UNET D2 Z Tol= 0.01
UNET D2 Volume Tol= 0.01
UNET D2 Max Iterations= 20
UNET D2 Equation= 0
UNET D2 RampUpFraction=0.1
UNET D2 TimeSlices= 1
UNET D2 Turbulence Formulation=Non-Conservative (original)
UNET D2 Eddy Viscosity=0.3
UNET D2 Transverse Eddy Viscosity=0.1
UNET D2 Smagorinsky Mixing=0
UNET D2 BCVolumeCheck=0
UNET D2 Cores=0
UNET D2 SolverType=PARDISO (Direct)
UNET D2 Minimum Iterations= 2147483647
UNET D2 Maximum Iterations= 2147483647
UNET D2 Restart Number= 10
UNET D2 Relaxation Coeff=1.3
UNET D2 SOR Precondition Iterations= 10
UNET D2 ILUT Maximum Fill= 8
UNET D2 ILUT Tolerance=1E-08
UNET D1D2 MaxIter= 0
UNET D1D2 ZTol=0.01
UNET D1D2 QTol=0.1
UNET D1D2 MinQTol=1
Write IC File= 0
Write IC File at Fixed DateTime=0
Write IC File at Sim End=0
Echo Input=False
Echo Parameters=False
Echo Output=False
Write Detailed= 0
HDF Write Warmup=0
HDF Write Time Slices=0
HDF Flush=0
HDF Compression= 1
HDF Chunk Size= 1
HDF Spatial Parts= 1
HDF Use Max Rows=0
HDF Fixed Rows= 1
Calibration Method= 0
Calibration Iterations= 20
Calibration Max Change=0.05
Calibration Tolerance=0.2
Calibration Maximum=1.5
Calibration Minimum=0.5
Calibration Optimization Method= 1
WQ AD Non Conservative
WQ ULTIMATE=-1
WQ Max Comp Step=1HOUR
WQ Output Interval=15MIN
WQ Output Selected Increments= 0
WQ Output face flow=0
WQ Output face velocity=0
WQ Output face area=0
WQ Output face dispersion=0
WQ Output cell volume=0
WQ Output cell surface area=0
WQ Output cell continuity=0
WQ Output cumulative cell continuity=0
WQ Output face conc=0
WQ Output face dconc_dx=0
WQ Output face courant=0
WQ Output face peclet=0
WQ Output face adv mass=0
WQ Output face disp mass=0
WQ Output cell mass=0
WQ Output cell source sink temp=0
WQ Output nsm pathways=0
WQ Output nsm derived pathways=0
WQ Create Restart=0
WQ Fixed Restart=0
WQ System Summary=0
WQ Write To DSS=0
Sorting and Armoring Iterations= 10
XS Update Threshold= 0.02
Bed Roughness Predictor= 0
Hydraulics Update Threshold= 0.02
Energy Slope Method= 1
Volume Change Method= 1
Sediment Retention Method= 0
Sediment TS Multiplier= 1
Warm Up Method= 0
XS Weighting Method= 0
Number of US Weighted Cross Sections= 1
Number of DS Weighted Cross Sections= 1
Upstream XS Weight=0
Main XS Weight=1
Downstream XS Weight=0
Number of DS XS's Weighted with US Boundary= 1
Upstream Boundary Weight= 1
Weight of XSs Associated with US Boundary= 0
Number of US XS's Weighted with DS Boundary= 1
Downstream Boundary Weight= 0.5
Weight of XSs Associated with DS Boundary= 0.5
Percentile Method= 0
Sediment Output Level= 3
Mass or Volume Output= 0
Output Increment Type= 1
Profile and TS Output Increment= 1
Transport Output Increment 1
XS Output Flag= 0
XS Output Increment= 10
Read HDF5 Sediment Hotstart= 0
Sediment Hotstart Type= 0
Write Gradation File= 0
Read Gradation Hotstart= 0
Write HDF5 File= 1
Write Binary Output= 1
Write DSS Sediment File= 0
DSS Sediment Output Type= 1
SV Curve= 0
Specific Gage Flag= 0
Subcell Erosion Methods= 0
Subcell Deposition Methods= 0
Advection Scheme= 1
Matrix Solver= 0
Implicit Weighting Factor= 1
Maximum Outer Loop Convergence Iterations= 5
Convergence Maximum Absolute= 0.001
Convergence RMSE= 0.0001
Grain Fractions Max Abs Error= 0.001
Max Subgrid Regions= 1
Max Subgrid Length Scale= 3.402823E+38
Initial Layer Thickness= 3.402823E+38
Min Layer Thickness= 3.402823E+38
Max Layer Thickness= 3.402823E+38
Number of Layers= 5

--- VALLEYFK.f01 (steady flow) ---

Flow Title=Flow
Program Version=6.20
Number of Profiles= 1
Profile Names=P100yr
River Rch & RM=VALLEYFK,Main            ,11954
     971
River Rch & RM=VALLEYFK,Main            ,9986
    1200
River Rch & RM=VALLEYFK,Main            ,7226
    1430
River Rch & RM=VALLEYFK,Main            ,6247
    1600
Boundary for River Rch & Prof#=VALLEYFK,Main            , 1
Up Type= 0
Dn Type= 3
Dn Slope=0.01731
DSS Import GetInterval= 0
DSS Import GetPeak= 0
DSS Import FillOption= 0

--- VALLEYFK.g01 (geometry) ---

Geom Title=Geometry
Program Version=6.20

River Reach=VALLEYFK        ,Main
Reach XY= 30
     2222115.939      560933.764     2221782.038      561016.536
     2221581.715      561143.179     2221281.593      561118.814
      2221077.08      561204.925     2220285.066      560943.467
 2220003.7629719561029.069268394      2219461.31      561021.794
     2219279.886      560911.551     2219124.276      560679.356
     2218691.916      560713.105     2218594.506      560744.135
     2218364.434      561058.758     2217554.805      561517.715
     2217089.782      561577.7842216833.83033608561483.683282813
2216645.25146564561605.186130226     2215909.661      561780.041
     2215362.539      561752.547     2214872.296      561399.379
     2214535.662      561394.073     2214253.966      561262.657
     2213579.799      561162.8532213159.06302816 560963.68331243
      2212802.89      560601.221     2212582.838      560653.739
     2212058.251      560526.536     2211890.116      560565.437
     2211548.786      560812.447     2211386.769      560736.893

Type RM Length L Ch R = 1 ,11954   ,280.9,281.5,281.1
XS GIS Cut Line= 4
2221921.10088019560454.6083333922222021.52286492560772.162083642
2222108.41507758 561056.807920222222256.68862714561296.978951876
#Sta/Elev= 30
       0 2747.18    23.7 2732.73    40.5 2717.78   107.6 2676.64   146.5 2657.45
   162.1 2645.51   178.9 2644.06   187.3 2639.29   199.9 2627.67     225 2625.66
   262.8 2610.72   304.8 2581.43   334.1 2573.65   384.3 2579.26   405.2  2578.3
   421.9 2572.59   472.1 2577.13     493 2575.92  500.62 2572.55   518.1 2571.97
   522.3 2572.53   537.9 2577.76   627.6 2577.19   691.1  2637.1   701.6 2644.81
     758 2667.76   772.1 2670.99   813.9 2691.64   828.2 2694.54   912.9 2737.05
#Mann= 6 ,-1,0
       0      .1       0     200     .06       0     310      .1       0
  500.62    .045       0   522.3     .06       0  613.05      .1       0
Bank Sta=500.62,522.3
XS Rating Curve= 0 ,0
Exp/Cntr(USF)=0,0
Exp/Cntr=0.3,0.1

Type RM Length L Ch R = 1 ,11673   ,187.2,187.6,185.2
XS GIS Cut Line= 4
2221655.23080086 560467.187677332221757.74990596560827.732395241
2221844.64211862561112.3782318192222117.57782373561372.355400337
#Sta/Elev= 30
       0 2753.97    76.6 2723.02   114.4 2703.22   126.8 2691.86   147.6 2690.42
   164.2 2680.67   222.5 2657.74   238.7 2643.14   267.9 2641.66   276.5 2638.36
   297.3 2623.78     310 2622.01   384.3  2578.4   422.4 2566.01   447.4 2566.52
     460 2570.18   476.7 2564.23   543.6 2565.46  551.542562.127   556.2 2561.59
  572.692562.171   610.6 2566.44   726.4 2568.18   765.7 2601.94   814.1 2629.99
   862.2 2650.23   931.4 2671.16   992.2 2703.85  1003.3 2706.62  1049.4 2729.57
#Mann= 7 ,-1,0
       0      .1       0     290     .06       0  394.84      .1       0
  551.54    .045       0  572.69      .1       0  712.45     .06       0
  752.45      .1       0
Bank Sta=551.54,572.69
XS Rating Curve= 0 ,0
Exp/Cntr(USF)=0,0
Exp/Cntr=0.3,0.1

Type RM Length L Ch R = 1 ,11485   ,244.2,251.2,258.2
XS GIS Cut Line= 3
       2221494.2        560657.6     2221655.505      561106.715
     2221887.444      561493.795
#Sta/Elev= 30
       0 2705.83    16.9 2690.68    29.3 2682.06    76.1 2655.07   110.7 2652.34
   132.6 2641.26   156.8 2631.68   169.6 2630.27   237.6  2595.6   275.8 2567.53
   288.6 2560.16   297.1 2557.59   331.1 2555.48   348.3 2559.24   407.7 2561.47
   432.7 2558.21   450.1 2559.42   461.72555.337   471.3 2554.03  483.532555.336
     497 2558.38   512.7 2567.11   546.6 2567.11   569.9 2569.61   595.2 2578.05
   634.2 2583.75   691.8 2597.72   741.2 2607.38   834.5 2640.39   928.5 2662.83
#Mann= 7 ,-1,0
       0      .1       0      90     .06       0     200      .1       0
   461.7    .045       0  483.53      .1       0   517.2     .06       0
   627.2      .1       0
Bank Sta=461.7,483.53
XS Rating Curve= 0 ,0
Exp/Cntr=0.3,0.1

Type RM Length L Ch R = 1 ,11234   ,308.3,306.4,302.2
XS GIS Cut Line= 4
2221390.96603592560704.8533009242221432.08556689561022.144721866
2221391.65387488561271.9918442792221398.95756313 561582.62338454
#Sta/Elev= 30
       0 2704.11     8.4 2702.11    40.7 2685.59    60.8 2666.73   101.2 2662.96
   113.3 2655.28   129.4 2652.23   141.5 2645.27   165.6 2642.61     202 2628.45
   229.9 2614.63   274.6 2586.88   286.7 2583.46   294.8 2576.67   306.9 2560.83
   318.7    2554   347.3 2548.88  411.452547.855   424.3 2546.85  441.072547.855
     469 2552.81   570.2  2550.9   586.2 2557.67   618.2 2580.95   633.3 2588.21
   698.3 2598.23   714.3 2609.04   822.3 2648.08   870.3 2667.05   883.8 2675.26
#Mann= 6 ,-1,0
       0      .1       0      40     .06       0     140      .1       0
  411.45    .045       0  441.07     .06       0  633.04      .1       0
Bank Sta=411.45,441.07
XS Rating Curve= 0 ,0
Exp/Cntr(USF)=0,0
Exp/Cntr=0.3,0.1

Type RM Length L Ch R = 1 ,10927   ,204,205.3,206.4
XS GIS Cut Line= 4
2221236.61556796560712.7925994292221145.20488929561017.468638686
2221130.51227431561232.0099645142221123.92490698561574.799017582
#Sta/Elev= 30
       0 2683.72    17.1 2680.91    74.5 2655.12   192.5 2626.94   259.3 2592.69
   284.4 2575.36   309.4 2553.06   321.8    2547   369.9 2542.57   426.1 2542.88
   446.1 2539.34   482.2 2542.54  493.532537.892   510.2 2536.72  515.272537.887
   526.3 2542.62   554.3 2544.53   566.3 2553.44   582.3 2569.11   630.3 2589.98
   650.3  2601.6   690.3 2604.92   706.3 2615.65   718.3 2619.99   730.3 2627.44
   758.3 2629.11   778.4 2640.94   802.4 2647.35   830.4 2661.02     876 2666.99
#Mann= 6 ,-1,0
       0     .06       0     140      .1       0  493.53    .045       0
  515.27      .1       0  543.14     .06       0  733.14      .1       0
#XS Ineff= 2 , 0
             475    2570
Permanent Ineff=
       F       F
Bank Sta=493.53,515.27
XS Rating Curve= 0 ,0
Exp/Cntr=0.3,0.1

Type RM Length L Ch R = 1 ,10722   ,101.2,99.6,98.4
XS GIS Cut Line= 4
2221068.68552308560736.863845278 2220949.4319182561074.181184813
2220922.17395137561221.8285051492220858.89041402 561594.32405713
#Sta/Elev= 30
       0 2656.61    59.7  2639.5    97.9 2631.53   114.9 2623.65   127.6 2622.37
   182.4 2593.43   208.2 2582.58   233.7 2565.74   246.4 2554.42   276.1  2541.3
   322.8 2538.67     344 2539.42   393.4 2534.08     437 2537.03  449.752531.446
   466.6 2530.42  476.572531.447   486.9 2535.55   511.3 2537.32   551.9 2576.64
   641.2 2626.41   653.3 2635.23     698 2640.31   718.2 2640.48   739.3 2649.45
   746.6 2654.73   762.9 2691.52   766.9 2695.29   815.6  2723.8   885.8 2753.91
#Mann= 5 ,-1,0
       0      .1       0  427.78     .06       0  449.75    .045       0
  476.57     .06       0  557.92      .1       0
Bank Sta=449.75,476.57
XS Rating Curve= 0 ,0
Exp/Cntr(USF)=0,0
Exp/Cntr=0.3,0.1

Type RM Length L Ch R = 1 ,10622   ,131.9,136,139.5
XS GIS Cut Line= 5
2220973.81182894 560739.769297182220843.82199235 561068.46971199
2220837.17598267561085.744500764 2220827.6045747 561221.35927474
2220776.70461919561578.603965914
#Sta/Elev= 30
       0 2642.52    60.9 2627.49    76.3 2621.33    91.5 2619.23   169.3 2588.84
   190.4 2579.03     251 2558.48     294 2537.68   395.5 2535.61  440.262528.542
   447.6 2527.43  461.18 2528.54   467.7 2531.68     496 2531.83   503.7 2534.77
   511.8 2540.77   535.6 2563.95   544.1 2575.08   564.3 2593.44   649.2 2640.36
   665.3 2642.92   713.8 2642.93   717.9 2645.17     734 2671.52   742.1 2682.19
   750.2 2689.65   782.5 2709.05     835 2735.45   851.2  2739.5   868.8 2748.94
#Mann= 5 ,-1,0
       0      .1       0  421.98     .06       0  440.26    .045       0
  461.18     .06       0  527.93      .1       0
Bank Sta=440.26,461.18
XS Rating Curve= 0 ,0
Exp/Cntr(USF)=0,0
Exp/Cntr=0.3,0.1

Type RM Length L Ch R = 1 ,10486   ,246.2,243.9,240.5
XS GIS Cut Line= 5
2220868.38346714560722.9209229032220718.89139558561086.759348327
2220710.00903317561104.1660221132220656.61876353561222.068788208
2220649.99930506561595.203890854
#Sta/Elev= 30
       0 2632.48      37 2621.55      50  2620.4   145.1 2592.27   158.1 2591.75
   176.6 2585.98   244.6 2561.64   261.9 2553.66   279.2 2540.99   286.9 2537.78
   326.8 2534.91   387.3 2533.63  404.292524.204   418.1 2523.17   428.62524.205
   440.4 2530.12   519.4 2527.02     537 2528.05   541.3 2530.01   565.5 2549.11
   581.4 2566.97     593 2572.84   673.5 2627.74   701.5  2640.6   765.5 2645.26
   769.5 2648.21   777.5 2663.17   781.5 2667.73   809.5 2687.62   915.5  2747.4
#Mann= 5 ,-1,0
       0      .1       0  404.29    .045       0   428.6      .1       0
  452.89     .06       0  562.32      .1       0
#XS Ineff= 2 , 0
                          469.45            2570
Permanent Ineff=
       F       F
Bank Sta=404.29,428.6
XS Rating Curve= 0 ,0
Exp/Cntr=0.3,0.1

Type RM Length L Ch R = 1 ,10243   ,257.1,256.1,253
XS GIS Cut Line= 4
2220573.24638616 560670.573787422220484.65799396560999.940886632
2220443.49923295561192.9467335422220468.46783568561580.422336995
#Sta/Elev= 30
       0 2614.45   168.4 2570.18   221.7 2547.26   263.7 2537.61   296.8 2524.78
   354.6 2521.61  371.782517.091   387.3 2515.89  396.582517.093   403.7 2523.98
   426.8  2520.6   493.7 2521.92   514.4 2519.25   534.6 2523.99   550.7  2533.6
   594.8 2549.72   622.8 2562.31   632.2 2569.72   642.9 2572.17   674.9 2592.06
     695 2610.71     719 2614.24   747.1 2635.43   771.1 2638.63   791.2 2650.09
   810.4  2655.5   827.2 2669.15   855.3 2673.28   871.3 2690.37   926.7 2721.47
#Mann= 5 ,-1,0
       0      .1       0  371.78    .045       0  396.58      .1       0
  481.07     .06       0  588.42      .1       0
#XS Ineff= 2 , 0
                          456.86            2550
Permanent Ineff=
       F       F
Bank Sta=371.78,396.58
XS Rating Curve= 0 ,0
Exp/Cntr(USF)=0,0
Exp/Cntr=0.3,0.1

Type RM Length L Ch R = 1 ,9986    ,270.8,268.3,265
XS GIS Cut Line= 4
2220269.63006304560663.2906299542220247.08765586560900.588941244
2220239.21488944561019.2972481472220295.82229521561594.022161877
#Sta/Elev= 30
       0 2626.74    53.8 2610.77    70.2  2602.7    82.3    2601   158.6  2573.4
   170.7 2565.85   190.7 2542.74   222.9 2519.68     239 2513.76   260.5 2512.87
  266.442509.782     283 2508.78  292.392509.779   319.1 2512.47   347.2 2510.57
   359.2 2514.77   415.5 2520.69   455.7 2520.14   467.7 2528.02     488 2528.16
   499.9  2533.2   556.2 2543.86   668.7  2589.6   684.8 2592.37   781.3 2631.28
   821.5  2655.6   861.6 2689.05   890.5 2692.01     926 2720.46   934.8 2723.48
#Mann= 5 ,-1,0
       0      .1       0  266.44    .045       0  292.39      .1       0
  477.34     .06       0  577.34      .1       0
Bank Sta=266.44,292.39
XS Rating Curve= 0 ,0
Exp/Cntr=0.3,0.1

Type RM Length L Ch R = 1 ,9718    ,222.7,224.5,226.6
XS GIS Cut Line= 4
2220093.46226511560673.3160228572219987.83764364560889.108260272
2220001.16887196561145.644426223 2220050.4742687561602.883650433
#Sta/Elev= 30
       0 2621.44    15.8 2620.39    26.6 2616.13    48.8 2618.38   111.2 2598.56
   169.1 2570.09   201.2 2534.89   225.1 2518.74   252.3 2506.11   276.4 2508.56
   304.4 2505.63   344.5 2506.13  375.182500.706   384.5 2499.26   393.62500.705
   404.5 2504.11   428.6 2502.39   464.6 2504.37   497.1 2514.41   516.8 2523.44
   573.1 2529.57   629.4 2548.36   657.6 2562.18   669.7 2565.03   681.7 2573.72
   731.9 2595.62   794.4  2626.9   919.1 2700.32   931.2 2711.04     957 2713.44
#Mann= 5 ,-1,0
       0      .1       0  375.18    .045       0   393.6      .1       0
  490.26     .06       0  587.14      .1       0
#XS Ineff= 2 , 0
                             405            2550
Permanent Ineff=
       F       F
Bank Sta=375.18,393.6
XS Rating Curve= 0 ,0
Exp/Cntr(USF)=0,0
Exp/Cntr=0.3,0.1

Type RM Length L Ch R = 1 ,9494    ,235.4,231.5,226.6
XS GIS Cut Line= 5
2220006.28745384560658.9495508172219792.88559541560890.428118453
      2219771.46      561015.2062219749.95569819561198.428407367
 2219929.8678552561606.927966356
#Sta/Elev= 30
       0  2613.2    93.7 2592.72   128.2  2578.2   175.7 2554.68   220.7 2537.42
   242.4 2518.61   258.7 2510.52   342.1 2505.34   419.1 2497.93  429.07 2494.44
   447.5 2493.18  454.192494.443   463.6 2496.92   499.8 2496.19   540.1 2499.35
   620.6 2497.72   628.9 2499.54   637.7 2504.98     657 2506.05   663.1 2509.75
   672.6 2519.16   702.5 2529.03   738.2 2536.62   760.2 2543.84   790.6 2559.47
   803.8  2562.4   945.3  2615.9  1026.7 2664.59  1052.9 2673.81  1072.3 2678.08
#Mann= 7 ,-1,0
       0      .1       0  429.07    .045       0  454.19      .1       0
  471.44     .06       0  571.44      .1       0  665.92     .06       0
  775.92      .1       0
Bank Sta=429.07,454.19
XS Rating Curve= 0 ,0
Exp/Cntr=0.3,0.1

Type RM Length L Ch R = 1 ,9262    ,202.7,209.6,218.1
XS GIS Cut Line= 4
2219542.74965524560673.4937688932219540.49008103560994.267563302
2219594.79933626561267.2819822942219459.30423356561574.740197375
#Sta/Elev= 30
       0 2562.11    75.7 2538.59   111.7 2531.01   167.7 2522.27   211.7  2518.8
   251.7 2496.74   319.7 2491.49  330.412488.344     340 2487.25  356.832488.343
   372.7 2490.33   387.6 2489.32   409.4  2492.4   474.7 2489.99   537.3  2490.2
   560.3 2492.92   572.5 2491.42   580.7 2495.26   601.2 2496.22   615.6 2500.93
   627.4 2505.08   644.9 2515.97   697.4 2523.59     730 2536.65     804 2574.11
   850.4 2595.11     881  2613.9   894.1 2624.33   902.8 2635.11   935.1 2659.05
#Mann= 5 ,-1,0
       0      .1       0  330.41    .045       0  356.83      .1       0
  570.78     .06       0  679.15      .1       0
Bank Sta=330.41,356.83
XS Rating Curve= 0 ,0
Exp/Cntr(USF)=0,0
Exp/Cntr=0.3,0.1

Type RM Length L Ch R = 1 ,9053    ,154.5,157.5,162
XS GIS Cut Line= 4
2219452.86776389560675.3301312212219360.66330215560950.779272443
2219176.91061974561224.2119649912219130.36668976561334.082597082
#Sta/Elev= 30
       0 2568.17    48.3 2550.67    86.3 2540.61   111.6 2536.48   145.4 2525.98
   153.8  2522.2   170.7 2520.42   179.1 2515.88   197.9 2510.19   213.7 2506.99
   271.9 2500.65   279.4 2496.38   293.4 2484.61   298.2 2482.13     303 2481.56
   312.2 2481.56     356 2483.31   373.3 2482.44   384.6 2479.56   399.2 2480.61
   413.3 2483.55   442.8 2483.79   592.2  2478.5   612.5 2479.58   638.3  2496.6
   652.6  2510.6     670 2530.12   680.6 2538.38   714.1  2553.8   739.2 2562.99
#Mann= 6 ,-1,0
       0      .1       0     303    .045       0   312.2      .1       0
  510.47     .05       0  520.47     .06       0  709.91      .1       0
#XS Ineff= 1 ,-1
  357.01  651.37 2515.09
Permanent Ineff=
       F
Bank Sta=303,312.2
XS Rating Curve= 0 ,0
Exp/Cntr=0.3,0.1

Type RM Length L Ch R = 1 ,8895    ,169.4,168.2,163.4
XS GIS Cut Line= 4
2219377.36305095560630.0626009562219265.41300017560841.359054426
2219105.89917614560935.8840723942218973.63909524561248.266283884
#Sta/Elev= 30
       0 2560.91    26.2 2549.96    94.1 2527.67   103.1  2523.1   118.6 2521.11
   133.4 2515.45   171.8 2505.96   233.2 2494.73   238.9 2491.43   245.7 2484.55
   254.5 2478.26   262.3 2476.56   283.7 2476.61   292.4  2479.4   319.6 2477.27
   339.2 2472.38   365.4 2477.61   429.9 2474.79   576.4 2472.32   588.6 2469.63
   595.4 2471.56   621.4 2471.63   625.8 2473.09   634.4 2479.45   652.7 2497.64
   667.9 2523.85     671 2527.91   695.4 2548.09   721.3 2563.43   763.8 2576.73
#Mann= 6 ,-1,0
       0      .1       0   262.3    .045       0   283.7      .1       0
  434.54     .05       0  534.54     .06       0  644.54      .1       0
#XS Ineff= 1 ,-1
  291.44   677.6 2519.84
Permanent Ineff=
       F
Bank Sta=262.3,283.7
XS Rating Curve= 0 ,0
Exp/Cntr(USF)=0,0
Exp/Cntr=0.3,0.1

Type RM Length L Ch R = 1 ,8727    ,298.1,297.2,290.5
XS GIS Cut Line= 4
2219283.31557606560574.120818915 2219179.8947733 560688.35171968
2218937.13417164561055.3206259622218924.69677521561244.070838146
#Sta/Elev= 30
       0 2555.24    22.6 2544.08    40.4  2532.2    55.4 2530.33     100  2509.5
   123.3 2500.52   153.7 2492.07   159.9 2485.96     166 2475.91  173.222471.244
   188.7 2471.31   209.3 2473.89   241.4 2473.76   255.5 2469.09   265.4  2468.6
   284.4 2472.57   303.8 2471.86   318.1 2476.39   332.5 2473.91   414.1 2473.16
   509.5 2467.76   559.6  2468.3   570.1 2466.76   596.7 2468.47     608 2472.94
   644.1 2508.14   676.1 2544.54   696.2 2556.36   728.2 2564.79   783.3 2573.52
#Mann= 5 ,-1,0
       0      .1       0  173.22    .045       0   188.7      .1       0
  454.09     .06       0  584.09      .1       0
#XS Ineff= 1 ,-1
  224.41  680.51 2550.55
Permanent Ineff=
       F
Bank Sta=173.22,188.7
XS Rating Curve= 0 ,0
Exp/Cntr(USF)=0,0
Exp/Cntr=0.3,0.1

Type RM Length L Ch R = 1 ,8430    ,247.1,246.2,244.6
XS GIS Cut Line= 4
2218900.86801773560458.4286115312218891.34229468560676.845664961
2218869.81629545560998.7397180362218895.76409643 561243.04290589
#Sta/Elev= 30
       0 2536.66    26.3 2525.71    70.8 2510.76   170.9 2488.41   190.9 2479.55
   206.9 2470.49     227 2462.53     251 2463.78  263.492461.673   275.1  2460.4
  281.52 2461.64   287.1 2463.41   308.3 2464.72   355.3 2464.58   395.4 2467.58
   467.5 2466.05   491.6 2462.66   515.6 2462.75   523.6 2460.36   543.7 2466.45
   567.8 2466.69   583.9 2473.89   608.1 2493.76   616.1 2502.69   624.1 2515.95
   632.2  2521.4   652.3 2530.16   724.7 2558.04   764.9 2567.21   786.9 2569.78
#Mann= 5 ,-1,0
       0      .1       0  263.49    .045       0  281.52      .1       0
  488.62     .06       0  581.24      .1       0
#XS Ineff= 1 ,-1
  316.21  644.08 2516.68
Permanent Ineff=
       F
Bank Sta=263.49,281.52
XS Rating Curve= 0 ,0
Exp/Cntr=0.3,0.1

Type RM Length L Ch R = 1 ,8184    ,264.1,258.9,253.6
XS GIS Cut Line= 4
2218552.51156315560486.1150538272218634.98625575560672.744836394
2218681.21384956560921.2947158622218863.37369491 561243.72537032
#Sta/Elev= 30
       0  2581.8    23.3 2577.56    44.5 2570.22    77.9 2552.11    95.2 2538.17
   117.1 2524.23   125.8 2520.95     132 2515.23   153.7 2504.12   208.6 2454.58
   241.1  2455.3   249.2 2453.69  259.182453.732   281.8 2457.71   302.1 2455.62
   315.2 2457.67   363.2  2458.1     377 2454.51   387.6 2455.87   403.8 2451.69
     448 2458.82   530.2 2458.27     547 2462.57   576.2 2461.99   611.6 2475.22
   655.6 2507.28   677.2 2518.34     737 2535.75   773.7 2551.65   827.2 2565.23
#Mann= 5 ,-1,0
       0      .1       0   249.2    .045       0  259.18      .1       0
  476.85     .06       0  596.85      .1       0
#XS Ineff= 1 ,-1
  316.94  353.37 2474.62
Permanent Ineff=
       F
Bank Sta=249.2,259.18
XS Rating Curve= 0 ,0
Exp/Cntr(USF)=0,0
Exp/Cntr=0.3,0.1

Type RM Length L Ch R = 1 ,7925    ,197,201.6,206
XS GIS Cut Line= 4
2218267.88656177560693.6462519762218424.07357993560878.865795963
2218547.80850201560953.0290080582218817.30470224561262.023898446
#Sta/Elev= 30
       0    2586    43.9 2576.36    74.9 2562.94    90.7 2559.09     137 2529.06
   151.1 2516.77   177.3 2500.11   195.7 2484.97   229.6 2461.05   242.4 2448.32
   249.9  2446.8   284.4 2447.81  294.85 2444.29   312.4 2443.18  324.272444.289
     331 2446.59   397.4 2450.69   411.4 2453.48   439.8 2454.73   460.6 2452.21
   492.9 2456.72   519.4 2456.14   534.3  2460.7   554.2 2460.47   620.3 2479.01
   681.7 2511.24     734 2536.01     747 2536.36   761.1 2543.05   796.5 2553.02
#Mann= 5 ,-1,0
       0      .1       0  294.85    .045       0  324.27      .1       0
  546.54     .06       0  696.54      .1       0
#XS Ineff= 2 , 0
          280.87 2459.82
Permanent Ineff=
       F       F
Bank Sta=294.85,324.27
XS Rating Curve= 0 ,0
Exp/Cntr=0.3,0.1

Type RM Length L Ch R = 1 ,7723    ,223.6,224.4,226.3
XS GIS Cut Line= 4
2218132.58080627560781.6734938682218299.46116049560995.076594232
2218383.67028622561103.1072820712218637.43560514561371.291075651
#Sta/Elev= 30
       0 2607.19    12.3 2602.64    25.3 2595.12    42.1  2592.4    70.6 2577.76
    90.8 2574.11   136.5 2554.79   148.7 2547.28   156.8 2539.73   167.5 2533.57
   202.5 2506.88   227.9  2486.8   241.6 2473.38   253.3 2468.96   258.7 2462.93
   270.1 2445.59   275.8 2440.24   329.4 2442.21  351.942438.156   363.2 2436.82
  374.152438.154   432.3 2449.16   474.8 2449.53   537.4  2453.5   573.8 2452.45
   610.6 2453.74   636.1 2466.11   689.8 2501.26   746.4 2535.44   777.1 2549.39
#Mann= 5 ,-1,0
       0      .1       0  351.94    .045       0  374.15      .1       0
  587.88     .06       0  727.88      .1       0
#XS Ineff= 2 , 0
          326.42 2455.81
Permanent Ineff=
       F       F
Bank Sta=351.94,374.15
XS Rating Curve= 0 ,0
Exp/Cntr(USF)=0,0
Exp/Cntr=0.3,0.1

Type RM Length L Ch R = 1 ,7499    ,271.3,272.6,275.9
XS GIS Cut Line= 5
2218064.39546871560830.1628476552218133.94417108561138.164243874
     2218158.959      561176.0212218212.98709504561267.931487883
2218448.93813521561534.070362296
#Sta/Elev= 30
       0 2602.89    48.2 2583.58    60.5 2575.39    76.9 2573.46    89.2 2567.66
   109.4 2565.08   122.8 2560.47   142.5 2550.68   154.8 2548.95   195.8 2520.27
   212.2 2507.03   256.6 2480.36   261.4 2476.26   277.8 2457.22   293.4 2455.18
   314.7 2438.74   319.8 2437.43   333.8 2438.94   342.6 2434.48  357.662430.886
   365.8 2429.81  383.162430.885   390.3 2435.03     395 2435.63   514.8 2438.87
   606.9 2445.27   624.4 2458.08   720.7 2505.07     768 2532.51   823.4 2554.63
#Mann= 5 ,-1,0
       0      .1       0  357.66    .045       0  383.16      .1       0
  537.75     .06       0  687.75      .1       0
Bank Sta=357.66,383.16
XS Rating Curve= 0 ,0
Exp/Cntr=0.3,0.1

Type RM Length L Ch R = 1 ,7226    ,173.8,173.1,166.6
XS GIS Cut Line= 4
2217886.92709992560917.1472990782217887.04751731561220.026525116
2217953.28437671561392.2423595612218367.83999787561597.981341309
#Sta/Elev= 30
       0 2577.42      32 2564.75      76 2551.53    85.2  2545.1     104 2542.32
     128 2526.87     144 2520.77     188 2497.18     208 2482.87     236 2477.55
     252 2465.39     264 2459.69   285.2 2440.86   310.8  2425.3     377 2428.65
   385.5  2427.3  391.052423.508   403.7 2422.14  417.892423.508   424.1 2427.11
   432.7 2428.01   463.1 2426.93   711.1 2435.91   727.3 2438.64   731.8 2439.87
   749.6 2453.58   773.8 2458.48   812.6 2471.32   874.7 2498.28   950.2 2535.64
#Mann= 7 ,-1,0
       0      .1       0  391.05    .045       0  417.89      .1       0
  577.39     .06       0  717.39      .1       0  797.39     .06       0
  827.39      .1       0
#XS Ineff= 2 , 0
          370.52 2442.54
Permanent Ineff=
       F       F
Bank Sta=391.05,417.89
XS Rating Curve= 0 ,0
Exp/Cntr(USF)=0,0
Exp/Cntr=0.3,0.1

Type RM Length L Ch R = 1 ,7053    ,163.4,164.2,165.5
XS GIS Cut Line= 4
2217726.40561013560952.2121478022217717.92817928561302.934317027
2217806.34195322561438.5304211152218331.59855502561610.476095884
#Sta/Elev= 30
       0 2548.66      33 2541.64      73 2529.28      85 2524.48      93 2519.15
     109 2517.85     133    2503     145 2501.68     157 2494.64     177 2492.25
     197 2479.44     253 2456.56     277 2453.05   309.1 2444.96   358.3 2421.67
   403.2 2423.45  418.442420.067   425.1 2419.17  452.022420.065     461 2423.59
   472.9 2421.12   508.7 2421.94   628.3 2428.01   741.9 2429.84     885 2437.51
   889.2 2438.34   905.6 2450.42   956.6 2466.03  1043.3 2504.99  1065.4 2516.44
#Mann= 5 ,-1,0
       0      .1       0  418.44    .045       0  452.02      .1       0
  510.82     .06       0   992.7      .1       0
#XS Ineff= 2 , 0
             400    2470
Permanent Ineff=
       F       F
Bank Sta=418.44,452.02
XS Rating Curve= 0 ,0
Exp/Cntr=0.3,0.1

Type RM Length L Ch R = 1 ,6889    ,296,297.5,298.4
XS GIS Cut Line= 6
2217498.64357742 561056.831807732217540.35947164561229.722096464
2217582.36146469561376.8993025632217671.75854887561544.418162997
2217685.95659829561649.4256643482217698.91711049561799.004489495
#Sta/Elev= 30
       0 2488.29    12.7 2479.92    33.3 2476.43    78.5 2478.66   119.7 2472.16
   160.8 2475.72     248  2447.7   302.1 2419.93   349.4  2420.8   367.5 2415.89
   403.8 2418.06   415.2 2415.14   428.2 2415.16   441.8 2413.18   456.6 2417.51
   489.9  2413.2     508 2419.08   541.7 2419.59   553.8    2437   561.9 2443.34
     574 2447.37   586.1 2464.98   598.2 2475.79   639.7 2499.97   670.7 2521.36
   682.7 2523.63   690.7 2531.46   734.9 2556.34   761.6 2576.36   776.9 2581.59
#Mann= 5 ,-1,0
       0      .1       0  400.91     .06       0   415.2    .045       0
   428.2     .06       0  510.91      .1       0
#XS Ineff= 2 , 0
          404.08 2423.49
Permanent Ineff=
       F       F
Bank Sta=415.2,428.2
XS Rating Curve= 0 ,0
Exp/Cntr=0.3,0.1

Type RM Length L Ch R = 1 ,6591    ,88.7,88.7,88.6
XS GIS Cut Line= 3
2217267.13985328561124.029175022 2217380.2944881561641.044660953
2217460.46454553561950.631746329
#Sta/Elev= 30
       0 2508.54    23.6 2497.25   122.8  2468.2   136.3 2461.62   148.6 2460.47
   242.8 2427.97   271.4 2415.34   351.4 2411.73   406.6 2412.57   410.6 2412.27
  418.32 2406.76   431.8  2405.2  443.35 2406.76   455.7 2412.05     513 2409.36
   537.7 2431.32   550.1 2436.03   595.5 2477.64   627.7    2497     641 2502.39
   660.5  2516.5     674 2520.66   682.3 2527.22   711.2 2541.27   756.6 2573.28
   773.2  2578.4   788.5  2590.9   818.6 2608.35   839.3 2616.61   849.1 2622.55
#Mann= 5 ,-1,0
       0      .1       0  418.32    .045       0  443.35      .1       0
     520     .06       0  619.25      .1       0
#XS Ineff= 2 , 0
                          455.69            2450
Permanent Ineff=
       F       F
Bank Sta=418.32,443.35
XS Rating Curve= 0 ,0
Exp/Cntr(USF)=0,0
Exp/Cntr=0.3,0.1

Type RM Length L Ch R = 1 ,6502    ,249.9,255.8,262.2
XS GIS Cut Line= 4
2217208.14257719561126.9830462722217239.69600875561414.136605611
2217291.85944575561650.3584814142217373.73885931561967.968601918
#Sta/Elev= 30
       0  2509.5     6.2  2509.1    34.4 2497.82   121.7 2475.98   147.1 2467.75
   155.1 2463.11   167.2 2461.49   199.4 2450.52   215.5  2443.1   263.8 2411.85
   279.9 2410.09   324.8 2412.01   357.5 2407.94     419 2407.27  434.282404.536
   444.7 2403.21  458.192404.537   468.1 2409.92   517.3 2406.42   529.6 2409.18
     542 2429.62   554.4  2434.4   570.9  2452.4   603.9 2476.91   674.2 2520.23
   686.5 2524.03     765  2575.4   779.7 2579.29   789.8 2588.55   858.8 2631.41
#Mann= 5 ,-1,0
       0      .1       0  434.28    .045       0  458.19      .1       0
  508.88     .06       0  610.79      .1       0
#XS Ineff= 2 , 0
                          472.24            2440
Permanent Ineff=
       F       F
Bank Sta=434.28,458.19
XS Rating Curve= 0 ,0
Exp/Cntr=0.3,0.1

Type RM Length L Ch R = 1 ,6247    ,216,214,203.5
XS GIS Cut Line= 4
2217129.53011109561131.5623548432217070.98252311561404.382043193
2217016.89545061561573.9177613322217115.22663518561983.461557772
#Sta/Elev= 30
       0 2499.88   125.4 2464.81   157.1 2452.99   173.5 2452.02   230.8    2437
     279 2415.15   309.3 2410.69   384.8 2404.28   397.4 2399.86     410 2400.45
  426.632398.076   435.2 2396.61  450.152398.077   456.2 2402.12   460.3  2402.6
   583.7 2403.32   596.1 2412.72   608.4 2417.78     629 2435.27   674.7 2467.96
   715.4 2489.31   727.7 2498.12     736 2500.79   768.9 2522.46   781.2 2525.58
   793.5 2535.73   826.5 2557.13   855.3 2580.67   867.6 2584.24   878.2 2592.91
#Mann= 5 ,-1,0
       0      .1       0  309.03     .06       0  426.63    .045       0
  450.15     .06       0  616.99      .1       0
Bank Sta=426.63,450.15
XS Rating Curve= 0 ,0
Exp/Cntr(USF)=0,0
Exp/Cntr=0.3,0.1

Type RM Length L Ch R = 1 ,6033    ,197.4,173,140.3
XS GIS Cut Line= 4
2216801.22865788561187.0962620952216824.83557703561473.091847668
2216869.17766431561754.5586178632217000.82451084562002.510313137
#Sta/Elev= 30
       0 2526.83    30.6  2514.8    46.2 2505.78    58.3 2503.39    98.4  2480.8
   130.5  2465.8   178.4 2448.97   186.7 2448.47   194.7 2443.61   206.8 2441.69
   230.9 2429.81   249.4 2427.26   264.2 2422.35     279 2411.88   291.1 2393.54
  293.642392.552   307.1 2391.28  319.782392.552   331.6 2395.82     364  2397.7
   477.4 2396.77   497.6 2398.36   521.9 2396.51   574.9 2400.47   595.4    2410
   608.6 2420.84   661.8 2453.43   715.3  2480.6   751.5 2504.41   852.6 2550.39
#Mann= 6 ,-1,0
       0      .1       0  293.64    .045       0  319.78      .1       0
  346.97     .06       0  446.97     .05       0  546.97      .1       0
Bank Sta=293.64,319.78
XS Rating Curve= 0 ,0
Exp/Cntr=0.3,0.1

Type RM Length L Ch R = 1 ,5860    ,100.9,107.8,110.2
XS GIS Cut Line= 4
2216580.72335038561268.4604493362216621.47709579561571.081834161
2216777.31455186561590.5353964472216860.97038228561873.919521989
#Sta/Elev= 30
       0 2501.19      29 2487.27    57.2 2471.31    81.4 2459.31    89.5 2453.93
   105.7 2450.65   113.7 2446.65   158.1 2431.42   170.2 2426.18   186.4 2423.48
   214.6 2412.08   222.7 2406.61   234.9 2394.92   275.2 2392.52   327.6 2393.07
   345.5 2387.57   354.6 2386.58   399.42388.411   413.6 2393.38     429 2395.39
   494.4 2396.58   519.4 2394.84   544.4 2394.91   594.4 2396.15   611.1 2398.29
   661.2 2400.75   669.5 2405.25     682 2416.38   714.8  2440.6   757.9 2466.17
#Mann= 7 ,-1,0
       0      .1       0     270     .06       0   345.5    .045       0
   399.4      .1       0   482.4     .06       0   502.4     .05       0
   612.4      .1       0
Bank Sta=345.5,399.4
XS Rating Curve= 0 ,0
Exp/Cntr(USF)=0,0
Exp/Cntr=0.3,0.1

Type RM Length L Ch R = 1 ,5752    ,233.5,259.5,277.7
XS GIS Cut Line= 5
2216512.33287705561258.8448118282216564.05678434561614.579749094
2216777.09281338561643.6834918892216815.74909417561822.621846725
2216927.65345308562044.800889402
#Sta/Elev= 30
       0 2501.89    34.7 2487.04    50.9 2477.93      63 2474.14    87.2 2459.04
    99.4 2457.47   114.8 2448.12   139.5  2436.2   168.1 2425.27   216.6  2410.9
   224.7 2406.32   240.8 2393.39   248.9 2389.81     257 2388.18   297.4 2388.46
   333.8 2390.51     350  2388.8   365.4 2385.03   386.8 2383.92   411.6 2385.21
     440  2390.5   604.7 2396.23   649.7 2395.49   678.3 2398.54   723.3 2400.15
   782.8 2440.52   858.1 2488.23   890.3 2504.23   975.4 2541.78  1006.3  2557.8
#Mann= 6 ,-1,0
       0      .1       0     280     .06       0   365.4    .045       0
   411.6     .06       0  594.49     .05       0  664.49      .1       0
Bank Sta=365.4,411.6
XS Rating Curve= 0 ,0
Exp/Cntr(USF)=0,0
Exp/Cntr=0.3,0.1

Type RM Length L Ch R = 1 ,5492    ,240.8,239.7,238
XS GIS Cut Line= 4
2216350.27715188 561218.25974309 2216309.1986139561474.289398223
2216350.00142662561707.5787259012216492.70839353562103.409517986
#Sta/Elev= 30
       0 2504.43    55.6 2484.33    91.7 2467.94   100.2 2461.17   112.3 2459.31
   144.7 2440.22   189.4 2420.18   233.9  2405.7   245.3 2398.55   262.2 2382.84
   283.8 2381.14   420.6 2383.27   428.7 2382.95  436.292379.462   447.6 2378.35
  465.732379.462   506.3  2386.2   585.1 2386.31   672.2 2391.52   676.4 2392.98
   691.2 2404.87   705.4 2413.18   714.7 2416.75   727.4 2418.45     746 2426.82
   765.7 2438.76   836.6 2486.59   850.8 2491.14   883.5 2513.02   916.9  2530.9
#Mann= 8 ,-1,0
       0      .1       0   319.3     .06       0   419.3     .05       0
  436.29    .045       0  465.73     .05       0  626.13      .1       0
  726.13     .05       0  896.13      .1       0
Bank Sta=436.29,465.73
XS Rating Curve= 0 ,0
Exp/Cntr=0.3,0.1

Type RM Length L Ch R = 1 ,5253    ,292.7,295.8,303
XS GIS Cut Line= 4
2216093.13611165561234.4688736952216054.16607792561509.181477925
2216140.13235308561831.4411443262216152.76336475 562121.00327297
#Sta/Elev= 30
       0 2480.19    99.7 2453.05   204.5 2417.73   237.5  2400.2   257.3  2382.4
   277.5 2376.44   318.9 2374.53   327.1  2372.5   343.7 2375.51   426.5  2378.2
   471.5 2377.75   492.7 2377.05  499.67  2373.6   517.4 2372.41  526.96 2373.69
   534.1 2378.02     588 2378.17   612.8 2383.62   652.8  2415.4   688.8 2441.17
   700.8 2444.76   736.8 2469.91   748.9  2473.7   756.9  2479.7   780.9  2492.3
   819.9 2516.13     845 2534.22     857 2537.64   869.7 2547.88   900.8 2567.19
#Mann= 5 ,-1,0
       0      .1       0  307.46     .06       0  407.46      .1       0
  499.67    .045       0  526.96      .1       0
Bank Sta=499.67,526.96
XS Rating Curve= 0 ,0
Exp/Cntr(USF)=0,0
Exp/Cntr=0.3,0.1

Type RM Length L Ch R = 1 ,4957    ,147,146.3,146.9
XS GIS Cut Line= 4
2215885.51160743561241.7917512682215859.99880986561491.918586342
2215821.26902193561803.7594772022215810.89220064562135.631251796
#Sta/Elev= 30
       0 2461.69   135.7 2427.49   168.3 2416.01   176.3 2414.85   208.5 2400.23
   226.2    2389   240.6 2377.32   252.7 2370.92   277.5 2371.08     293 2369.23
   349.4 2371.84   389.7  2371.8   397.8 2373.24   409.9 2370.41   442.1 2365.93
   502.6 2370.04   522.8 2369.34   528.5 2366.69  555.512366.921   567.1 2375.39
   579.1 2379.02   591.1 2389.96     599 2395.04   643.1 2414.63   687.1 2424.03
   783.2 2439.24   815.2 2446.98   831.2 2449.32   847.2 2449.59   897.7 2462.12
#Mann= 5 ,-1,0
       0      .1       0  291.42     .06       0  391.42      .1       0
   528.5    .045       0  555.51      .1       0
#XS Ineff= 2 , 0
           397.8    2400
Permanent Ineff=
       F       F
Bank Sta=528.5,555.51
XS Rating Curve= 0 ,0
Exp/Cntr=0.3,0.1

Type RM Length L Ch R = 1 ,4810    ,121.1,120.8,124.3
BEGIN DESCRIPTION:
structure xs 4
END DESCRIPTION:
XS GIS Cut Line= 4
2215768.09526419561241.7325831522215690.86435816561489.325781882
2215676.43257975561827.1918311012215702.81132142562139.790303384
#Sta/Elev= 30
       0  2452.9    34.6 2444.09    83.2 2428.81   124.1 2427.48   175.9 2410.24
   200.7 2397.97   225.7 2379.88   242.4 2370.15   258.2  2365.2   339.3 2369.02
   399.3 2367.28   415.4 2364.13   435.4 2366.78   523.5 2365.45   531.5 2363.98
  582.242365.525   595.5 2374.43   611.6 2376.54   619.6 2381.73   631.6 2392.63
   651.7    2406   663.8 2411.94   675.8  2420.8   702.8 2435.05     724 2448.36
     740 2452.95   752.1 2461.92   779.7 2476.48   812.3 2487.07   911.2 2511.94
#Mann= 9 ,-1,0
       0      .1       0     200     .06       0     240     .08       0
  299.36     .06       0  399.36      .1       0   523.5    .045       0
  582.24      .1       0  697.53     .05       0  857.53      .1       0
#XS Ineff= 2 , 0
          338.59    2385
Permanent Ineff=
       F       F
Bank Sta=523.5,582.24
XS Rating Curve= 0 ,0
Exp/Cntr(USF)=0,0
Exp/Cntr=0.3,0.1

Type RM Length L Ch R = 1 ,4690    ,50.8,50.3,50.2
BEGIN DESCRIPTION:
structure xs 3
END DESCRIPTION:
XS GIS Cut Line= 4
2215673.07812077561233.3869431422215581.36726523561466.954863299
2215550.49642606561867.0255470392215551.07323608562120.383193266
#Sta/Elev= 30
       0 2448.94    56.1 2433.73    68.5 2428.82    85.7 2427.68    98.6 2422.58
   171.7 2404.06   188.9 2398.27   197.5 2393.63   214.6 2375.53     232 2363.71
   289.3 2363.86   309.3 2366.08   349.4 2366.36   365.5 2368.77   395.5 2364.32
   453.8 2364.13   489.9 2359.37   518.5 2362.52  545.072361.937   566.1 2361.95
   602.2 2361.01   614.2 2367.04   622.3 2368.29   682.3 2388.82   696.8 2398.61
   722.3 2419.29   767.8 2445.15   806.3 2470.46   878.3 2521.79   905.5 2538.32
#Mann= 5 ,-1,0
       0     .05       0     220     .08       0  320.93     .05       0
  545.07    .045       0   566.1     .05       0
#XS Ineff= 2 , 0
          530.07  2363.7   581.1            2365
Permanent Ineff=
       F       F
Bank Sta=545.07,566.1
XS Rating Curve= 0 ,0
Exp/Cntr(USF)=0,0
Exp/Cntr=0.3,0.1

Type RM Length L Ch R = 1 ,4639    ,156.9,160.3,167.7
BEGIN DESCRIPTION:
structure xs 2
END DESCRIPTION:
XS GIS Cut Line= 4
2215622.71749732561234.7877947832215531.00664178 561468.35571494
2215500.13580261 561868.426398682215500.71261263562121.784044907
#Sta/Elev= 30
       0 2441.49    32.7  2432.7    45.5 2426.89    65.5  2424.6    88.5 2417.46
   114.3  2415.9   148.7 2400.25     192 2372.83   217.4 2363.92   279.8 2363.48
   309.6 2364.92   396.2 2362.47   436.3 2363.38   460.4 2362.72   484.4 2358.52
   496.4 2358.18   536.6 2361.79   547.7  2358.9  558.86  2358.9   580.7 2358.23
   592.8  2359.5   656.9 2377.08     677 2385.45   696.9 2396.16   724.9 2416.87
   760.9 2439.98   804.9    2472   813.3 2476.58   872.9 2517.98   905.5 2535.98
#Mann= 6 ,-1,0
       0     .05       0     220     .08       0  320.93     .05       0
   547.7    .045       0  558.86     .05       0  640.93      .1       0
#XS Ineff= 2 , 0
           542.3  2363.7  564.26            2365
Permanent Ineff=
       F       F
Bank Sta=547.7,558.86
XS Rating Curve= 0 ,0
Exp/Cntr(USF)=0,0
Exp/Cntr=0.3,0.1

Type RM Length L Ch R = 1 ,4479    ,202.6,207.4,212.3
BEGIN DESCRIPTION:
structure xs 1
END DESCRIPTION:
XS GIS Cut Line= 6
2215542.41124282561188.7460992092215509.33843737561281.749234561
2215419.32358415561549.0880430282215363.71049724561706.698055279
2215338.83256268561779.1634496042215269.64914832562113.560071825
#Sta/Elev= 30
       0 2432.53    30.2  2424.4    98.1 2425.22   114.9 2422.76   144.5 2412.25
   165.5 2408.35   177.6 2403.79   187.6 2398.27   224.7 2370.38   233.2 2370.77
   266.9 2361.88   339.1 2362.75     421 2357.66   482.7 2361.12   503.9  2357.7
   516.6 2359.31   533.6 2355.89   562.1 2357.59  570.952355.613   605.5 2354.52
  618.712355.613   628.5 2364.45   638.9 2368.51   657.4 2389.63   671.5 2401.59
   732.8 2416.66   822.7 2433.19   909.4 2455.12   945.2 2460.81     966 2466.49
#Mann= 6 ,-1,0
       0     .05       0  128.71      .1       0  258.71     .06       0
  430.79      .1       0  570.95    .045       0  618.71      .1       0
#XS Ineff= 2 , 0
          516.63    2375
Permanent Ineff=
       F       F
Bank Sta=570.95,618.71
XS Rating Curve= 0 ,0
Exp/Cntr=0.3,0.1

Type RM Length L Ch R = 1 ,4272    ,278.4,279.9,284.3
XS GIS Cut Line= 4
2215424.38299892561138.1919734262215299.94049932561323.737975831
2215152.77477173561698.4355345132214935.17385028561976.334398714
#Sta/Elev= 30
       0 2424.96    57.8  2412.7    75.8 2405.73   129.6 2396.97   151.2 2388.51
   178.2 2386.34   210.7  2362.2   227.4 2357.85   319.5    2355   388.3 2357.86
   474.3 2356.66   508.6 2352.98   521.5 2347.72   547.3 2351.37   554.5 2349.61
   569.9 2349.61   588.4 2349.91     616 2354.68   649.8 2374.66   702.4 2419.69
   716.7 2423.86     726 2433.89   753.7 2456.14   807.3 2489.24   870.5 2535.96
   887.6 2539.56   904.7 2555.76   930.4 2569.64   944.6 2580.03   978.9 2597.27
#Mann= 5 ,-1,0
       0      .1       0  233.41     .06       0  453.41      .1       0
   554.5    .045       0   569.9      .1       0
Bank Sta=554.5,569.9
XS Rating Curve= 0 ,0
Exp/Cntr(USF)=0,0
Exp/Cntr=0.3,0.1

Type RM Length L Ch R = 1 ,3992    ,208.8,200.6,195.2
XS GIS Cut Line= 5
2215297.72241835561061.4264732972215185.80109665561237.830925019
     2214960.408      561469.1872214897.33269178561541.527948892
2214825.77768683561901.173458713
#Sta/Elev= 30
       0 2433.39    93.7 2408.53   103.9 2402.25   127.6 2400.79   144.8 2391.56
   171.9 2382.43   189.3 2368.94   208.1 2359.07   223.7 2355.62   308.5 2349.94
     409 2349.37   447.2 2345.23   461.4 2347.71     501 2346.63  509.842342.531
   529.2 2341.54   543.4 2342.41   550.5 2344.48   622.1  2343.6     652  2366.7
   664.2 2383.47   676.2 2395.89     717 2425.87   725.4 2431.53   741.7 2435.95
   888.6 2532.74   904.9 2535.48   917.1 2543.82   941.5 2552.78   994.6 2565.29
#Mann= 5 ,-1,0
       0      .1       0  348.91     .06       0  468.91      .1       0
  509.84    .045       0   543.4      .1       0
#XS Ineff= 2 , 0
          472.73 2351.73
Permanent Ineff=
       F       F
Bank Sta=509.84,543.4
XS Rating Curve= 0 ,0
Exp/Cntr=0.3,0.1

Type RM Length L Ch R = 1 ,3791    ,258.2,259.2,258.6
XS GIS Cut Line= 4
2214951.49350907560922.7614815572214880.58261174561110.219177903
2214746.21866039561496.8005490132214630.66487931561876.232919739
#Sta/Elev= 30
       0 2431.08    77.2 2383.97   105.2 2375.39   118.1 2373.65   143.7 2360.52
   159.6 2354.62   175.1 2352.85   190.8 2344.02   254.4 2340.54     301 2343.33
   347.9 2341.79   423.8 2343.68   466.1 2340.95  472.512337.967  501.912338.124
   512.7 2339.95   538.1 2336.72   559.3 2341.44   597.4 2340.89   622.6 2348.34
     677 2388.67   697.9 2406.91   714.6  2416.2   775.5    2432   794.1 2433.54
   806.6 2439.37   863.8 2452.95   877.7 2458.63   911.1 2465.14  1006.3 2492.39
#Mann= 5 ,-1,0
       0      .1       0  340.42     .06       0  440.42      .1       0
  472.51    .045       0  501.91      .1       0
#XS Ineff= 2 , 0
          421.86 2367.97
Permanent Ineff=
       F       F
Bank Sta=472.51,501.91
XS Rating Curve= 0 ,0
Exp/Cntr(USF)=0,0
Exp/Cntr=0.3,0.1

Type RM Length L Ch R = 1 ,3532    ,240.3,238.5,237.4
XS GIS Cut Line= 4
2214746.09819466560863.5952696512214589.95601056561234.538911403
 2214524.6775602561408.8105176622214401.80916294  561820.2557801
#Sta/Elev= 30
       0 2409.79   118.7 2363.95   131.9 2362.45   179.8  2333.4   225.6 2333.12
   244.8 2338.36   271.5 2339.07   465.1 2333.53   524.9 2336.14  559.76 2332.25
   576.1 2330.76  589.12 2332.25   601.5 2344.89     615 2350.54   618.2 2354.48
   626.5 2372.49   643.2 2391.28     660 2397.05   668.3 2406.03   680.8  2414.2
   722.5 2430.99   760.1 2453.89   772.6 2455.77   789.3 2470.49     806 2472.85
   831.1 2487.54   878.6 2509.08   893.7 2510.61   953.8  2534.9    1018 2570.67
#Mann= 5 ,-1,0
       0      .1       0     300     .06       0  402.47      .1       0
  559.76    .045       0  589.12      .1       0
#XS Ineff= 2 , 0
          524.89    2355
Permanent Ineff=
       F       F
Bank Sta=559.76,589.12
XS Rating Curve= 0 ,0
Exp/Cntr=0.3,0.1

Type RM Length L Ch R = 1 ,3293    ,285.6,281.9,277.7
XS GIS Cut Line= 4
2214467.61507909560742.7537622342214452.85034705 560873.36485331
2214302.93152947561331.0715463832214211.93136452561762.333036177
#Sta/Elev= 30
       0 2416.76   106.6 2363.47   123.2 2360.62     173 2337.67   215.4 2327.57
   282.8 2326.24   358.5 2333.72   417.5 2333.43   430.1 2327.97   496.4 2326.95
   518.5 2331.99   539.5 2331.05  550.752326.097   560.6 2324.62  590.132326.098
   602.7 2329.95   613.8 2340.46   623.4 2344.75   656.1 2379.03   667.8 2387.78
     759 2434.06   795.1 2458.65   811.5  2461.9   827.8  2475.1   889.1 2509.99
   900.7 2513.19   921.8 2531.56   934.1 2534.06   966.8 2558.53  1053.8 2609.61
#Mann= 5 ,-1,0
       0      .1       0  311.44     .06       0  411.44      .1       0
  550.75    .045       0  590.13      .1       0
#XS Ineff= 2 , 0
          514.28    2350
Permanent Ineff=
       F       F
Bank Sta=550.75,590.13
XS Rating Curve= 0 ,0
Exp/Cntr(USF)=0,0
Exp/Cntr=0.3,0.1

Type RM Length L Ch R = 1 ,3011    ,453.3,457.3,461.6
XS GIS Cut Line= 5
2214157.28827745560647.0170144452214080.66326385560787.139106083
 2214049.3738091561159.926704376  2214039.987357561261.163206492
2213997.27217441561742.808356661
#Sta/Elev= 30
       0  2410.2    61.4 2370.14    75.4 2354.58    89.1 2350.63   116.4 2327.61
   125.6 2323.21   165.8 2319.78   306.3 2320.92   326.3 2317.15   386.5 2322.63
   462.8 2319.78   486.9 2325.99   575.2  2324.1  598.632318.566  626.382318.536
   659.6 2337.46   667.6 2354.56   671.6 2358.92   710.6 2387.21   731.9 2393.51
   751.9 2405.92     764 2409.19   782.9 2422.35   800.1 2425.87   819.7 2439.82
   872.4  2467.8   884.5 2469.39   900.5 2481.72   976.8 2523.05    1119 2590.64
#Mann= 5 ,-1,0
       0      .1       0   319.7     .07       0   419.7      .1       0
  598.63    .045       0  626.38      .1       0
#XS Ineff= 2 , 0
          571.22    2340
Permanent Ineff=
       F       F
Bank Sta=598.63,626.38
XS Rating Curve= 0 ,0
Exp/Cntr=0.3,0.1
